--- WHITEOAKCK.prj (project) ---

Proj Title=WHITEOAKCK
Current Plan=p01
Default Exp/Contr=0,0
English Units
Geom File=g01
Flow File=f01
Plan File=p01
BEGIN DESCRIPTION:
END DESCRIPTION:
DSS Export Rating Curves= 0
DSS Export Rating Curve Sorted= 0
DSS Export Volume Flow Curves= 0
DXF OffsetX= 0
DXF OffsetY= 0
DXF ScaleX= 0
DXF ScaleY= 0

--- WHITEOAKCK.p01 (plan) ---

Plan Title=Floodplain
Program Version=4.00
Geom File=g01
Flow File=f01
K Sum by GR=0
Std Step Tol=0.01
Critical Tol=0.01
Num of Std Step Trials=20
Max Error Tol=0.3
Flow Tol Ratio=0.001
Split Flow NTrial=30
Split Flow Tol=0.02
Split Flow Ratio=0.02
Log Output Level=0
Friction Slope Method=1
Unsteady Friction Slope Method=2
Unsteady Bridges Friction Slope Method=1
Global Log Level=0
CheckData=False
Run HTab=0
Run UNet=0
Run PostProcess=0
UNET Theta=0
UNET Theta Warmup=0
UNET ZTol=0
UNET ZSATol=0
UNET MxIter=0
UNET MaxInSteps=0
UNET DtIC=0
UNET DtMin=0
UNET MaxCRTS=0
UNET WFStab=0
UNET SFStab=0
UNET WFX=0
UNET SFX=0
UNET DSS MLevel=0
UNET DZMax Abort=0
UNET Convert EG Bridges=0
UNET Use Existing IB Tables=0
UNET Froude Limit=0
UNET Froude Power=0
Write IC File=0
Echo Input=False
Echo Output=False
Write Detailed=0

--- WHITEOAKCK.f01 (steady flow) ---

Flow Title=NFF Regression Equation
Program Version=4.10
Number of Profiles= 1
Profile Names=P100yr
River Rch & RM=WHITEOAKCK,Main            ,29805.5
 1203.16
River Rch & RM=WHITEOAKCK,Main            ,25692.4
1338.975
River Rch & RM=WHITEOAKCK,Main            ,24798.1
 1766.99
River Rch & RM=WHITEOAKCK,Main            ,18991.4
1887.897
River Rch & RM=WHITEOAKCK,Main            ,18072
3063.933
River Rch & RM=WHITEOAKCK,Main            ,14523.1
3274.366
River Rch & RM=WHITEOAKCK,Main            ,7266.9
3668.294
Boundary for River Rch & Prof#=WHITEOAKCK,Main            , 1
Up Type= 0
Dn Type= 3
Dn Slope=0.004
DSS Import GetInterval= 0
DSS Import GetPeak= 0
DSS Import FillOption= 0

--- WHITEOAKCK.g01 (geometry) ---

Geom Title=USGS 10m DEM
Program Version=4.10

River Reach=WHITEOAKCK      ,Main
Reach XY= 30
     1821876.555      374072.443     1820745.881      375157.641
       1820299.7      375391.039     1819546.228      376543.817
     1818606.124      377360.657     1818252.825      378313.782
     1817842.235      378822.029     1817466.367      380423.331
     1817442.929      381620.119     1816837.894      382639.216
     1815912.113      383040.475     1814121.749      382033.313
      1812672.53      381630.319     1812457.686      381752.715
     1811883.731      381628.102     1811171.228      381245.553
     1810352.217      381241.647     1809431.645      381558.053
     1809107.426      381931.751     1808750.655       385093.21
     1808292.564      385985.775     1807414.961      385976.661
     1807103.762       386113.38     1806417.804      386852.531
     1806060.143        386938.9     1805393.476      387506.348
     1804747.643      387817.546     1804112.226      387790.203
     1803703.372      387515.463     1803157.799      387731.608

Type RM Length L Ch R = 1 ,29805.5 ,129.1,130.2,131.4
XS GIS Cut Line= 3
     1821562.822      373809.076      1821869.94      374079.943
     1822177.059      374350.809
#Sta/Elev= 30
       0 1256.31    11.9 1245.81    19.9 1241.55    55.7 1238.67    63.6  1236.8
    67.6 1234.77   107.3 1200.03   135.2 1180.12     167 1169.52   210.7 1152.33
   242.5  1134.2   274.3 1131.68   337.9 1130.57   385.6 1126.79   405.5 1126.77
   417.4 1126.36   433.4 1126.76   481.1 1128.85   500.9 1131.25   508.9  1134.1
   564.6 1172.93   576.5 1178.91   604.3 1196.77     652 1230.67   671.9 1240.74
   707.7 1266.62   739.5 1292.14   755.4 1301.83   771.3 1308.56     819 1335.14
#Mann= 3 , 0 , 0
       0     .07       0   405.5    .045       0   433.4     .07       0
Bank Sta=405.5,433.4
XS Rating Curve= 0 ,0
Exp/Cntr=0.3,0.1

Type RM Length L Ch R = 1 ,29675.2 ,9.1,19.3,29.7
XS GIS Cut Line= 2
     1821526.256      373928.982      1822049.26      374433.539
#Sta/Elev= 30
       0 1229.98       8 1228.21      28 1229.58    35.9 1226.64    43.9 1221.28
    87.8 1184.76   107.8 1170.97   159.7 1140.12   195.6 1123.09   207.6 1120.47
   251.6 1116.27   331.4 1112.21   349.2 1107.85   363.4 1107.45   369.2 1107.72
   383.3 1111.08   423.2    1114   435.2  1118.4   451.2 1131.95   495.1 1162.53
     543 1191.62     595 1228.08   610.9 1236.72   618.9 1238.92   626.9 1242.78
   646.8 1257.87   662.8 1267.22   678.8 1280.71   694.8  1291.9   726.7 1310.84
#Mann= 3 , 0 , 0
       0     .08       0   349.2    .045       0   369.2     .08       0
Bank Sta=349.2,369.2
XS Rating Curve= 0 ,0
Exp/Cntr=0.3,0.1

Type RM Length L Ch R = 1 ,29655.9 ,40.2,40.1,40.2
XS GIS Cut Line= 4
     1821539.277      373946.994     1821755.206      374155.327
     1821793.183      374234.537     1822038.409      374449.381
#Sta/Elev= 30
       0 1228.81     7.9 1228.89    19.7 1223.48    63.2 1186.85    86.9 1169.94
   142.1 1137.59   157.9 1129.26   173.7 1122.62   185.6 1120.03   236.9  1115.5
     316  1112.3   333.3 1107.54     348 1106.79   353.3 1107.23   371.9  1110.5
   403.8 1112.16   411.8 1113.92   415.7  1115.8   427.6 1125.63   471.4  1158.3
   491.3 1171.84   546.9 1206.01   570.8  1225.9   586.7 1235.61   610.5 1245.78
   634.4 1263.64   646.3 1270.78   662.2 1282.47   682.1 1295.47   713.9 1313.61
#Mann= 3 , 0 , 0
       0     .08       0   333.3    .045       0   353.3     .08       0
Bank Sta=333.3,353.3
XS Rating Curve= 0 ,0
Exp/Cntr=0.3,0.1

Type RM Length L Ch R = 1 ,29615.8 ,80.3,67.9,54.7
XS GIS Cut Line= 4
     1821517.576      373981.716     1821733.504       374190.05
     1821771.482       374269.26     1822016.707      374484.103
#Sta/Elev= 30
       0 1225.53     7.9 1223.68    11.8 1221.26    43.4 1194.83    90.8 1161.01
   138.2  1131.9     154 1124.44   169.8 1119.49   189.5 1116.49   209.2 1116.61
   244.8  1113.3     308 1110.82   331.7 1106.35     344 1105.81   351.7 1106.21
   367.9 1109.25   399.8 1111.33   407.8 1113.86   423.7 1128.63   455.5 1152.39
   483.3 1172.15     539 1208.98   550.9 1219.61   562.8 1227.97   590.7  1242.3
   618.5 1264.08   674.2  1298.9   690.1 1305.37     702 1312.54   713.9 1316.62
#Mann= 3 , 0 , 0
       0     .09       0   331.7    .045       0   351.7     .09       0
Bank Sta=331.7,351.7
XS Rating Curve= 0 ,0
Exp/Cntr=0.3,0.1

Type RM Length L Ch R = 1 ,29548   ,222.7,223.3,224
XS GIS Cut Line= 2
      1821426.43      374055.501     1821979.815      374493.869
#Sta/Elev= 30
       0 1213.89    23.9 1212.78    43.9 1200.13    75.8 1176.76    95.7 1168.96
   103.7 1164.19   147.6 1150.07   179.5 1128.07   199.4 1126.88   231.3 1121.75
   287.2 1117.54     339 1109.28   351.2  1105.7     363 1104.82   371.2 1105.59
   386.9 1107.79   410.8 1108.74   418.8 1110.94   454.7    1142   478.6 1158.16
   490.6 1167.72   514.5  1182.9   550.4 1208.15   578.3 1231.03   606.3  1246.3
   622.2 1259.85   650.1  1275.1   674.1 1291.29     686 1296.49     706  1307.6
#Mann= 3 , 0 , 0
       0     .09       0   351.2    .045       0   371.2     .09       0
Bank Sta=351.2,371.2
XS Rating Curve= 0 ,0
Exp/Cntr=0.3,0.1

Type RM Length L Ch R = 1 ,29324.7 ,176.2,189.8,203.4
XS GIS Cut Line= 2
     1821279.945      374206.326     1821813.799      374650.119
#Sta/Elev= 30
       0  1219.8      16 1208.99    27.9 1198.36    35.9 1192.62    43.9  1190.5
    67.8 1189.65    75.8 1186.36    87.8 1184.28   107.7 1175.28   127.7 1161.75
   143.6 1155.89   203.5 1126.81   215.4 1124.06   227.4 1124.13   251.4 1119.77
   311.2 1113.19   335.1 1100.41   339.1 1100.11   355.1 1100.25   367.1 1102.59
     411 1104.76   418.9 1106.26   458.8  1131.8   538.6 1174.72   582.5 1203.54
   602.5 1213.98   622.4 1219.92   650.3 1222.43   662.3  1222.1   694.2 1225.34
#Mann= 3 , 0 , 0
       0     .09       0   335.1    .045       0   355.1     .09       0
Bank Sta=335.1,355.1
XS Rating Curve= 0 ,0
Exp/Cntr=0.3,0.1

Type RM Length L Ch R = 1 ,29134.8 ,300.6,289.2,277.9
XS GIS Cut Line= 4
     1821109.589      374377.767     1821388.452      374472.168
     1821477.428      374709.798     1821779.077      374938.747
#Sta/Elev= 30
       0 1253.15    15.9 1245.51    51.7 1218.01    79.6 1203.37   107.4 1175.46
   115.4 1169.81   123.3 1167.12   151.2 1167.43   163.1 1163.33   234.7 1107.46
   242.7 1105.79   278.5 1105.37   298.4 1111.21     338 1099.01     346 1098.72
   421.3 1098.88   437.1 1099.62     449 1104.37     457 1105.55   472.8  1103.7
   556.1 1106.96     596 1114.36   727.5 1131.54   783.3  1140.4   807.3 1136.52
   863.1 1139.03     879 1141.86     895 1148.37   910.9 1149.99   926.8 1154.96
#Mann= 3 , 0 , 0
       0     .06       0     338    .045       0   421.3     .06       0
Bank Sta=338,421.3
XS Rating Curve= 0 ,0
Exp/Cntr=0.3,0.1

Type RM Length L Ch R = 1 ,28845.6 ,215.5,219,222.5
XS GIS Cut Line= 2
     1820996.742      374539.442     1821488.279      375028.808
#Sta/Elev= 30
       0 1231.03    63.8 1188.25    83.7 1171.92    95.7 1151.55    99.7 1147.32
   103.6 1144.67   107.6 1143.36   131.6 1141.52   143.5 1136.96   151.5 1131.47
   155.5 1127.18   163.4 1115.76   171.4 1108.06   179.4 1102.26   183.4 1100.44
   191.3 1099.03   406.6 1098.85   410.6 1098.97   418.6 1100.56   446.5 1112.79
   462.4  1113.8   470.4 1115.75   506.2 1130.58   526.2  1137.5   546.1 1147.18
   558.1 1154.96     566 1161.23   621.8 1196.56   653.7 1212.25   693.6  1240.5
#Mann= 3 , 0 , 0
       0     .05       0   191.3    .045       0   410.6     .05       0
Bank Sta=191.3,410.6
XS Rating Curve= 0 ,0
Exp/Cntr=0.3,0.1

Type RM Length L Ch R = 1 ,28626.6 ,143,140.2,137.5
XS GIS Cut Line= 2
     1820879.077       374675.64     1821221.959      375128.114
#Sta/Elev= 30
       0 1195.84      20 1181.36      40 1169.34      52 1157.47      60 1152.34
      68 1145.81      80 1138.22      88 1134.11     108 1134.38   111.9 1133.36
   115.9 1131.16   123.9 1122.86   147.9 1103.59   155.9 1100.02   163.9 1098.86
   355.8 1098.56   363.8  1098.7   379.8 1100.14   395.8 1104.08   411.8 1104.71
   419.8 1107.49   427.8 1113.48   455.8 1130.62   459.8 1132.59   475.8 1137.58
   483.8 1141.47   503.8 1155.11   519.7 1168.25   551.7 1191.92   567.7 1199.19
#Mann= 3 , 0 , 0
       0     .05       0   163.9    .045       0   363.8     .05       0
Bank Sta=163.9,363.8
XS Rating Curve= 0 ,0
Exp/Cntr=0.3,0.1

Type RM Length L Ch R = 1 ,28486.4 ,46.1,47.4,48.8
XS GIS Cut Line= 2
     1820706.378      374739.616     1821166.447      375226.812
#Sta/Elev= 30
       0 1209.16       8 1202.97    27.9 1190.44    55.8  1167.6    71.8 1157.68
    91.7 1139.16   103.7 1129.15   115.7 1122.48   119.7 1121.32   139.6 1121.37
   147.6 1119.31   175.5 1097.01   183.5 1092.57   203.4 1087.49   227.4 1084.28
   311.1 1084.03   324.7  1080.3     339 1079.64     347  1080.3     355 1082.01
     363  1086.1     367  1086.8   438.8 1089.44   442.7 1090.92   462.7  1107.5
   534.5 1150.51   582.3 1185.93   598.3 1193.62   654.1 1231.46   670.1 1240.16
#Mann= 3 , 0 , 0
       0     .09       0   324.7    .045       0     347     .08       0
Bank Sta=324.7,347
XS Rating Curve= 0 ,0
Exp/Cntr=0.3,0.1

Type RM Length L Ch R = 1 ,28439   ,130.6,133.1,135.3
XS GIS Cut Line= 2
     1820688.582      374764.051     1821104.164      375254.503
#Sta/Elev= 30
       0  1200.6      12 1191.12    31.9 1180.21    43.9 1169.69    59.9 1157.67
    79.9 1144.96    95.8 1128.12   103.8 1121.66   111.8 1118.64   131.8 1117.93
   139.8  1115.3   147.7 1109.99   163.7 1094.94   167.7 1093.05   215.6 1083.62
   311.4 1081.62   319.4 1079.09   331.4  1078.3   337.3 1078.72   351.4 1082.73
   367.3  1082.9   411.3 1086.57   427.2  1092.9   471.2 1121.89   495.1 1134.55
     527 1155.92     563 1182.21     583 1193.26   630.9 1226.92   642.8 1232.69
#Mann= 3 , 0 , 0
       0     .09       0   319.4    .045       0   337.3     .09       0
Bank Sta=319.4,337.3
XS Rating Curve= 0 ,0
Exp/Cntr=0.3,0.1

Type RM Length L Ch R = 1 ,28305.9 ,346.2,344.4,342.5
XS GIS Cut Line= 2
     1820589.841      374799.859     1821029.041      375427.181
#Sta/Elev= 30
       0 1212.97       4  1211.2    75.8 1163.06   111.7 1132.97   139.6 1112.47
   147.6 1107.89   175.5 1105.64   191.4 1094.25   211.4 1088.45   279.2 1081.51
     347 1081.14   356.4 1076.83   370.9 1075.78   376.4 1076.36   386.9 1079.92
   426.8 1081.24   434.7 1082.85   454.7 1096.96   474.6 1106.84   486.6 1115.37
   514.5 1131.36   542.4 1149.67   554.4 1155.58   590.3 1179.69   614.2 1189.95
   666.1 1223.41     706 1237.58   725.9 1249.06   741.9 1252.42   765.8 1266.61
#Mann= 3 , 0 , 0
       0      .1       0   356.4    .045       0   376.4      .1       0
Bank Sta=356.4,376.4
XS Rating Curve= 0 ,0
Exp/Cntr=0.3,0.1

Type RM Length L Ch R = 1 ,27961.5 ,96.8,87.8,78.9
XS GIS Cut Line= 2
     1820198.131       374900.77       1820730.9      375544.216
#Sta/Elev= 30
       0 1243.23      28 1227.75      40 1225.42      68 1213.24    87.9 1207.23
   119.9 1190.82   151.9  1184.1   163.9 1176.78   187.9 1171.72   203.8 1155.71
   235.8 1132.76   267.8 1114.95   299.8 1100.56   319.8    1084   327.8 1079.44
   359.7 1076.22   419.7 1076.56   451.7 1071.51   475.6 1072.44   487.6 1069.13
   499.6 1068.23   507.6 1069.42   567.6 1072.34   591.6 1091.32   643.5 1123.48
   675.5 1146.62   719.5 1175.16   735.5 1181.94   791.4 1215.12   835.4 1228.32
#Mann= 3 , 0 , 0
       0      .1       0   487.6    .045       0   507.6      .1       0
#XS Ineff= 2 , 0
       0   471.6 1072.86               0
Permanent Ineff=
       F       F
Bank Sta=487.6,507.6
XS Rating Curve= 0 ,0
Exp/Cntr=0.3,0.1

Type RM Length L Ch R = 1 ,27873.7 ,38.7,38,38
XS GIS Cut Line= 4
     1820060.327      374955.023     1820395.614      375300.076
     1820466.143      375343.478     1820674.477       375602.81
#Sta/Elev= 30
       0  1262.1    19.9 1249.24    35.8 1244.34    59.6 1231.81    71.6 1229.35
   131.2 1205.94     159 1190.36   214.7 1168.52   222.7 1163.04   254.5 1158.29
   318.1 1120.28   381.7  1076.3   417.5 1072.94     489 1070.93   512.7 1067.37
   532.4  1067.1   540.3 1067.18   563.9 1070.25   611.5 1071.53   635.2 1092.67
   651.1 1102.87   702.5 1130.29   738.2 1153.47   765.9 1173.79   785.7 1184.39
   821.3 1207.94   841.1 1218.61   860.9 1226.05   876.8 1229.62   896.6 1238.97
#Mann= 3 , 0 , 0
       0      .1       0   512.7    .045       0   540.3      .1       0
Bank Sta=512.7,540.3
XS Rating Curve= 0 ,0
Exp/Cntr=0.3,0.1

Type RM Length L Ch R = 1 ,27835.7 ,50.5,57.4,64.2
XS GIS Cut Line= 4
     1820037.541      374981.065     1820372.827      375326.117
     1820443.357       375369.52      1820651.69      375628.852
#Sta/Elev= 30
       0 1265.78    23.9 1252.53    75.6 1229.37    99.4 1224.58   135.2 1206.95
   147.1 1198.71     167 1194.97   206.8  1173.9   226.6 1156.42   254.5 1150.69
   278.3 1132.53   361.8 1083.52   385.7 1074.83   417.5 1070.94   465.2 1070.81
   508.7 1066.87   520.6  1066.3   528.4 1067.05   548.2 1070.55   599.6 1069.29
   607.5 1071.35   619.4 1083.43   643.1  1100.2   698.6 1132.96   761.9  1177.3
   773.8 1182.35   813.4 1208.59   833.2 1219.61     857 1226.04   896.6 1244.64
#Mann= 3 , 0 , 0
       0      .1       0   508.7    .045       0   528.4      .1       0
Bank Sta=508.7,528.4
XS Rating Curve= 0 ,0
Exp/Cntr=0.3,0.1

Type RM Length L Ch R = 1 ,27778.3 ,300,297.7,295.1
XS GIS Cut Line= 2
     1820053.817      375055.935     1820588.756      375616.916
#Sta/Elev= 30
       0 1242.46      24 1228.89      40 1226.06    67.9  1207.7    91.9 1199.05
   127.9 1171.64   139.8  1168.8   147.8 1164.63   171.8 1143.91   187.8 1140.61
   211.8 1122.12   295.7 1076.55   319.6 1069.88   395.6 1070.57   411.6 1066.59
   423.7  1065.9   435.5 1064.51   443.7 1066.06   459.5 1069.68   515.4 1067.28
   527.4 1068.16   535.4 1070.93   571.4  1098.3   627.3 1132.28   651.3 1148.97
   667.3 1162.35   679.3 1168.86   743.2 1212.42   759.2 1218.99   775.2 1221.24
#Mann= 3 , 0 , 0
       0      .1       0   423.7    .045       0   443.7      .1       0
#XS Ineff= 2 , 0
       0   395.6                       0
Permanent Ineff=
       F       F
Bank Sta=423.7,443.7
XS Rating Curve= 0 ,0
Exp/Cntr=0.3,0.1

Type RM Length L Ch R = 1 ,27480.5 ,475.8,469,461.4
XS GIS Cut Line= 2
     1819895.397      375341.308     1820407.549      375774.251
#Sta/Elev= 30
       0 1177.77    31.9 1158.97    95.8 1115.18   107.8 1112.15   127.7 1102.12
   147.7 1099.07   187.6 1087.31   203.6 1076.93   219.6 1073.93   235.5 1062.18
   267.4 1060.56   299.4  1064.6   331.3 1064.23   348.9 1058.26   363.3 1056.44
   371.2 1057.62   395.2 1063.82   407.2 1062.89   415.2 1065.18   431.1 1079.98
     471 1109.05     491 1114.27     507 1123.24   526.9 1140.74   578.8 1176.62
   594.8  1183.5   626.7 1205.26   638.7 1209.12   654.7 1210.62   670.6 1219.61
#Mann= 3 , 0 , 0
       0      .1       0   348.9    .045       0   371.2      .1       0
#XS Ineff= 2 , 0
       0   323.3                       0
Permanent Ineff=
       F       F
Bank Sta=348.9,371.2
XS Rating Curve= 0 ,0
Exp/Cntr=0.3,0.1

Type RM Length L Ch R = 1 ,27011.5 ,382.3,389.2,396.3
XS GIS Cut Line= 2
     1819578.556      375774.251     1820171.004      376079.155
#Sta/Elev= 30
       0 1211.64       8 1212.24    43.9 1194.92    91.8 1162.74   103.7  1156.8
   151.6 1120.32   163.6 1108.33   179.5  1104.1   211.5 1083.82   223.4 1072.01
   231.4 1066.03   239.4 1056.59   247.4 1051.32   287.3 1048.09   319.2 1052.42
   359.1 1053.62     379 1049.46     399 1048.02     407 1046.61     421 1047.94
   442.9 1057.93   462.8 1056.28   474.8 1057.88   498.7 1069.48   526.7  1090.5
   542.6 1093.62   558.6 1106.46   598.5 1131.32   638.4 1162.73   666.3 1180.06
#Mann= 3 , 0 , 0
       0      .1       0     399    .045       0     421      .1       0
#XS Ineff= 2 , 0
       0   355.1                       0
Permanent Ineff=
       F       F
Bank Sta=399,421
XS Rating Curve= 0 ,0
Exp/Cntr=0.3,0.1

Type RM Length L Ch R = 1 ,26622.3 ,499.8,509.9,520.1
XS GIS Cut Line= 3
     1819418.414      376014.194     1819736.543      376272.255
     1820051.977      376533.427
#Sta/Elev= 30
       0 1225.23    19.9 1208.73    31.8 1206.52    71.6 1187.99   111.4 1158.09
   143.2 1138.78     171 1116.84   182.9  1105.4   198.8 1099.73   234.6 1080.97
   278.4 1046.79   290.3 1044.06   373.8 1044.23   396.6 1039.31   405.7 1038.54
   417.6 1039.47   429.5 1043.76   445.4 1045.81   524.9 1048.51   532.9 1051.24
   544.8  1063.1   552.8 1067.44   572.6 1074.45   592.5 1077.16   600.5 1082.29
   616.4 1087.74   656.1 1096.42   747.6 1107.73   791.3 1117.47   819.2 1119.44
#Mann= 3 , 0 , 0
       0      .1       0   396.6    .045       0   417.6      .1       0
Bank Sta=396.6,417.6
XS Rating Curve= 0 ,0
Exp/Cntr=0.3,0.1

Type RM Length L Ch R = 1 ,26112.4 ,429.7,419.9,409.5
XS GIS Cut Line= 2
     1819211.803      376287.489     1819534.069      376889.702
#Sta/Elev= 30
       0 1154.56      16 1143.89      32 1137.13    43.9 1129.94    83.9 1101.84
    87.9 1099.68    99.9 1097.18   115.8 1085.06   151.8 1066.52   179.7 1046.43
   187.7 1042.14   259.6 1035.61   279.6 1030.78   299.6 1034.38   323.5 1035.33
   351.5 1034.22   367.5 1028.93   375.5 1027.79   387.4  1029.5   399.4 1029.69
   419.4 1033.22   459.3 1033.62   463.3 1035.65   487.3 1060.73   507.3 1074.42
   563.2 1101.32   599.1 1124.18   615.1 1132.67     659 1150.02     683 1162.73
#Mann= 3 , 0 , 0
       0      .1       0   367.5    .045       0   387.4      .1       0
#XS Ineff= 2 , 0
       0   343.5                       0
Permanent Ineff=
       F       F
Bank Sta=367.5,387.4
XS Rating Curve= 0 ,0
Exp/Cntr=0.3,0.1

Type RM Length L Ch R = 1 ,25692.4 ,464.8,462.6,460.2
XS GIS Cut Line= 3
     1818918.834      376494.737     1818879.772      376731.282
     1819301.864      377070.909
#Sta/Elev= 30
       0 1092.96       8 1091.19      36 1077.71    67.9 1068.45   115.9 1041.37
   123.9 1037.78   139.8 1033.93   179.8 1030.04   207.8 1030.14   235.8 1026.61
   275.6 1025.87   303.5 1027.12   387.1 1023.91   407.1 1028.24   450.9 1027.16
   458.8  1023.5   466.8 1021.63   478.8 1020.77   490.7 1021.54   518.6 1027.28
   554.4 1057.43   578.4 1073.52   602.2 1086.13   626.2 1102.46     654 1124.89
     674  1136.6   717.8 1169.24   741.7 1177.31   757.6  1187.5   781.5 1200.15
#Mann= 3 , 0 , 0
       0      .1       0   466.8    .045       0   490.7      .1       0
#XS Ineff= 2 , 0
       0   407.1                       0
Permanent Ineff=
       F       F
Bank Sta=466.8,490.7
XS Rating Curve= 0 ,0
Exp/Cntr=0.3,0.1

Type RM Length L Ch R = 1 ,25229.8 ,437.6,431.7,426.5
XS GIS Cut Line= 2
     1818431.638      376987.359     1818993.704      377379.069
#Sta/Elev= 30
       0 1145.58    31.9 1128.76    71.7 1102.94    99.6 1081.46   119.5 1076.81
   143.4 1065.72   163.3 1055.87   215.1 1025.46     231 1022.97     243 1018.39
   278.8 1018.78   294.8  1015.2   306.7 1014.68   330.6 1018.86   350.5 1019.04
   374.4 1013.84   382.4 1012.68   394.4  1013.6   410.3 1016.59   430.2 1016.45
   446.1 1014.31   489.9 1016.66   497.9 1022.51   509.8 1035.88   521.8  1046.9
   557.6 1070.23   573.6 1082.12   581.5 1085.09   621.4  1115.8   685.1 1159.21
#Mann= 3 , 0 , 0
       0      .1       0   374.4    .045       0   394.4      .1       0
#XS Ineff= 2 , 0
       0   342.6                       0
Permanent Ineff=
       F       F
Bank Sta=374.4,394.4
XS Rating Curve= 0 ,0
Exp/Cntr=0.3,0.1

Type RM Length L Ch R = 1 ,24798.1 ,488.2,492.6,495.9
XS GIS Cut Line= 2
     1818239.581      377415.961     1818821.178      377700.249
#Sta/Elev= 30
       0  1121.5      20 1113.28    63.9 1087.71    71.9 1081.64    87.9 1065.13
    91.9 1062.42   107.9  1059.6   127.9 1043.13   155.8 1027.34   175.8 1018.74
   183.8 1013.16   199.8 1009.28   211.8    1008   239.8 1006.74   247.8 1007.24
   259.7 1010.64   291.7 1010.27     332 1004.62   339.7 1003.75     352 1004.29
   387.6 1008.72   435.6 1008.44   459.6 1009.74   463.5 1011.29   499.5 1040.95
   515.5 1052.29   539.5 1066.65   603.4 1110.93   635.4 1130.33   647.4 1139.31
#Mann= 3 , 0 , 0
       0      .1       0     332    .045       0     352      .1       0
#XS Ineff= 2 , 0
       0   267.7                       0
Permanent Ineff=
       F       F
Bank Sta=332,352
XS Rating Curve= 0 ,0
Exp/Cntr=0.3,0.1

Type RM Length L Ch R = 1 ,24305.5 ,361.9,364.5,367.8
XS GIS Cut Line= 3
     1817983.068      377799.321     1818340.125      377999.833
     1818696.131      378202.192
#Sta/Elev= 30
       0 1193.57    15.9 1184.79    39.8 1164.76    75.5 1141.24   107.4 1124.91
   119.3 1123.79   147.1 1104.75   194.8 1082.27   226.6 1056.64   242.5 1049.35
   270.4 1026.98   298.2 1000.92   310.1  998.05     330 1000.73   349.9  995.87
   361.8   999.7   393.6 1000.39   405.5  995.46   413.5  993.99   429.4  996.13
   453.2 1000.49   481.1  996.96   560.6    1009   580.5 1007.84   620.2  1021.2
     648 1022.73   727.6 1038.48   739.5 1042.79   775.3 1065.24     819 1078.38
#Mann= 3 , 0 , 0
       0      .1       0   405.5    .045       0   429.4      .1       0
#XS Ineff= 2 , 0
       0   393.6                       0
Permanent Ineff=
       F       F
Bank Sta=405.5,429.4
XS Rating Curve= 0 ,0
Exp/Cntr=0.3,0.1

Type RM Length L Ch R = 1 ,23940.9 ,358.2,360.7,361.2
XS GIS Cut Line= 2
     1817954.207      378119.086     1818432.723      378486.925
#Sta/Elev= 30
       0 1100.75      24 1088.66      64  1061.1    83.9 1045.11    99.9 1037.01
   115.9 1025.35   151.9  995.22   155.9  992.96   163.9  991.94   183.9  993.44
   195.9  990.96   203.8  990.79   215.8  993.37   247.8  993.86   275.8  988.07
   331.8  988.61   343.8  987.41   355.7  988.55   379.7  994.52   395.7  990.85
   403.7  990.74   431.7  999.93   435.7 1002.15   443.7 1010.56   459.7 1023.74
   523.6 1063.92   543.6 1079.17   555.6 1085.28   587.6  1097.2   603.6 1105.89
#Mann= 3 , 0 , 0
       0      .1       0   331.8    .045       0   355.7      .1       0
#XS Ineff= 2 ,-1
       0   247.8  993.86   379.7     500  994.52
Permanent Ineff=
       F       F
Bank Sta=331.8,355.7
XS Rating Curve= 0 ,0
Exp/Cntr=0.3,0.1

Type RM Length L Ch R = 1 ,23580.2 ,303.4,298,292.1
XS GIS Cut Line= 2
     1817667.749      378354.546     1818217.879      378726.725
#Sta/Elev= 30
       0 1117.07       8 1112.25    19.9 1110.43    35.8 1103.05    67.6 1085.17
    99.4 1072.65   131.2  1057.1   159.1 1037.88     171 1033.46   186.9 1030.64
   194.9 1027.63   242.6  999.09   258.5  987.85   306.2  985.25     346  988.57
   373.9  987.58   385.8  984.77   405.7  983.24   413.6  981.95   425.6   982.8
   441.5  984.25   461.4  983.42   485.2  985.41   501.1  989.23   513.1   995.9
     525 1006.21   572.7 1037.66   616.5 1071.98   624.4 1076.37   664.2 1090.43
#Mann= 3 , 0 , 0
       0      .1       0   405.7    .045       0   425.6      .1       0
#XS Ineff= 2 , 0
       0     342                       0
Permanent Ineff=
       F       F
Bank Sta=405.7,425.6
XS Rating Curve= 0 ,0
Exp/Cntr=0.3,0.1

Type RM Length L Ch R = 1 ,23282.2 ,327.9,324.6,321
XS GIS Cut Line= 2
     1817545.136      378702.853     1818113.713      378920.952
#Sta/Elev= 30
       0 1095.25    35.8 1076.43    59.7 1059.08    71.6 1048.67    87.6 1043.17
   107.5  1025.8   131.4    1018   175.1  984.15   183.1  979.88     195  978.48
   238.8  978.35   254.7  979.92   266.7  983.69   298.5  984.97   306.5  983.25
   314.4  979.14   318.4   977.9   334.3  979.78   342.3  981.01   358.2  979.39
   386.1  981.12   413.9  980.35   421.9   981.8   437.8  993.42   465.7 1010.53
   493.6 1030.86   513.4 1047.69   521.4  1052.4   589.1 1079.41     609 1085.48
#Mann= 3 , 0 , 0
       0      .1       0   314.4    .045       0   334.3      .1       0
#XS Ineff= 2 , 0
       0   294.5                       0
Permanent Ineff=
       F       F
Bank Sta=314.4,334.3
XS Rating Curve= 0 ,0
Exp/Cntr=0.3,0.1

Type RM Length L Ch R = 1 ,22957.5 ,440.1,436.6,432.8
XS GIS Cut Line= 2
     1817395.397      379029.459     1818045.353       379194.39
#Sta/Elev= 30
       0 1114.62      24 1101.32    39.9 1096.52    75.8 1078.44   107.8 1065.37
   119.7 1056.41   135.7 1050.16   167.6 1022.83   183.6 1016.33   207.6  998.01
   211.5  994.05   223.5  977.51   227.5  973.94   231.5  972.72   251.5  973.99
   299.4  973.39   319.3  976.77   343.3  976.73   355.2  972.14   367.2  970.27
   378.1  972.27   403.1   976.4     459  978.51     475  982.26   490.9  983.68
   526.9 1004.51   538.8 1014.06   590.7 1046.06   646.6 1072.79   670.6 1080.73
#Mann= 3 , 0 , 0
       0      .1       0   355.2    .045       0   378.1      .1       0
#XS Ineff= 2 , 0
       0   339.3             403       0
Permanent Ineff=
       F       F
Bank Sta=355.2,378.1
XS Rating Curve= 0 ,0
Exp/Cntr=0.3,0.1

Type RM Length L Ch R = 1 ,22520.9 ,370,375,380
XS GIS Cut Line= 2
     1817246.742      379505.805     1817932.506      379565.484
#Sta/Elev= 30
       0 1112.46    31.8 1091.36    47.8 1085.02    75.6 1064.22   103.4 1057.43
   127.3 1047.17   151.2 1034.37   175.1 1019.21   210.9 1001.53   222.8  993.38
   274.6  972.33   322.3  963.35   338.2  964.84   350.2  969.41   358.1  970.54
     382  970.71   392.5  965.77   401.9  962.46   412.5  965.14   449.6  965.84
   469.5  971.62   501.4  971.42   525.2  974.79   541.1   979.1     561  987.32
   604.8 1014.82   616.7  1019.6   652.6 1045.62   672.4 1052.54   688.4 1066.02
#Mann= 3 , 0 , 0
       0      .1       0   392.5    .045       0   412.5      .1       0
#XS Ineff= 2 , 0
       0     378                       0
Permanent Ineff=
       F       F
Bank Sta=392.5,412.5
XS Rating Curve= 0 ,0
Exp/Cntr=0.3,0.1

Type RM Length L Ch R = 1 ,22145.9 ,275.8,270.9,265.7
XS GIS Cut Line= 2
     1817191.404      379791.178     1817929.251      380010.362
#Sta/Elev= 30
       0 1087.85    31.9 1079.73    55.8 1065.07    71.8 1057.69    87.7 1046.41
   115.7 1041.39   139.6 1026.14   155.5 1010.34   179.5 1006.94   191.4 1002.94
   227.3  975.49   251.2  962.15   307.1  957.59     339  962.83   370.9  963.28
   386.8  958.85   394.8  956.32   410.8  957.93   434.7  958.79   454.6   962.8
   486.6  960.04   502.5  961.21   510.5  965.93   534.4  992.41   618.2    1051
   638.1 1060.46     662 1068.77   693.9 1085.64   737.8 1100.92   769.7 1120.46
#Mann= 3 , 0 , 0
       0      .1       0   386.8    .045       0   410.8      .1       0
#XS Ineff= 2 , 0
       0   366.9                       0
Permanent Ineff=
       F       F
Bank Sta=386.8,410.8
XS Rating Curve= 0 ,0
Exp/Cntr=0.3,0.1

Type RM Length L Ch R = 1 ,21875   ,444.9,445.3,445.4
XS GIS Cut Line= 2
     1817175.128        380138.4     1817844.615      380198.079
#Sta/Elev= 30
       0 1047.74    19.9 1040.58    47.7 1017.12    71.6 1002.07    83.5  999.36
   111.4  998.33   127.3   994.3     171  966.51   186.9  958.55   202.8  956.66
   222.7  957.49   234.6  954.36   254.5  953.22   266.5  953.64   278.4  956.74
   318.2  958.25   334.1  953.19     342  952.74   360.3  953.33   397.7   959.9
   433.5  978.76   477.3 1007.14   505.1 1032.62     517 1039.44   532.9 1044.95
   564.8 1049.41   580.7    1061   592.6  1073.4   660.2 1097.65   672.1 1103.15
#Mann= 3 , 0 , 0
       0      .1       0   334.1    .045       0   360.3      .1       0
#XS Ineff= 2 , 0
       0     318  958.24               0
Permanent Ineff=
       F       F
Bank Sta=334.1,360.3
XS Rating Curve= 0 ,0
Exp/Cntr=0.3,0.1

Type RM Length L Ch R = 1 ,21429.7 ,391.4,389.9,388.2
XS GIS Cut Line= 2
     1817102.428      380569.173      1817755.64      380634.277
#Sta/Elev= 30
       0 1048.48    27.8 1029.47    55.7  1026.4    63.7 1022.55    75.6 1008.47
    95.5   992.8   107.4  989.72   139.2  988.39   159.1  980.64   171.1  970.64
     183  965.48   206.9  962.22   222.8  956.12   238.7  953.74   254.6  946.87
   278.5  951.69   310.3  951.79   338.2  945.02   350.1  943.67     362  945.17
   405.8  949.39   453.6  950.26   477.4  956.86   501.3  972.15     545 1008.42
   600.8 1022.41   620.6 1035.24   636.6  1038.5   644.5 1045.38   656.4 1061.18
#Mann= 3 , 0 , 0
       0      .1       0   338.2    .045       0     362      .1       0
#XS Ineff= 2 , 0
       0     306   951.7               0
Permanent Ineff=
       F       F
Bank Sta=338.2,362
XS Rating Curve= 0 ,0
Exp/Cntr=0.3,0.1

Type RM Length L Ch R = 1 ,21039.8 ,482.1,484.4,487.4
XS GIS Cut Line= 2
     1817085.067      380970.648     1817827.254      380995.605
#Sta/Elev= 30
       0 1073.97      16 1065.85    35.9 1060.65    63.9 1040.66    79.8 1034.05
    99.8 1018.01   143.7 1011.52   159.7 1005.76   247.5  941.91   283.5  942.72
   327.4  939.06   359.3  945.12   371.3  944.05   383.8  938.77   391.3   937.1
   403.8  939.12   419.2  943.41   439.2  941.11   451.2  943.72     519  992.24
     531  997.98   614.8     997   638.8  1000.7   642.8 1002.33   646.8 1009.04
   650.8 1020.88   658.8 1035.55   674.7  1051.3   702.7 1064.68   742.6 1075.36
#Mann= 3 , 0 , 0
       0      .1       0   383.8    .045       0   403.8      .1       0
#XS Ineff= 2 , 0
       0   359.3   945.1               0
Permanent Ineff=
       F       F
Bank Sta=383.8,403.8
XS Rating Curve= 0 ,0
Exp/Cntr=0.3,0.1

Type RM Length L Ch R = 1 ,20555.5 ,487.9,500,509.6
XS GIS Cut Line= 3
     1817058.438       381410.82     1817465.889      381457.531
      1817869.71      381524.835
#Sta/Elev= 30
       0 1115.84    43.8 1087.45    79.6 1067.12    91.6 1061.78   123.4 1053.37
   191.1 1015.69     223 1000.97   238.9  987.26   258.8  980.84   290.7  952.24
   314.6  935.02   330.5  930.96   350.4  936.88   382.2  937.12   386.2   936.7
   398.2  929.57   410.1  927.69   420.1  929.42   441.9  936.29   469.7  932.96
   533.3   937.9     585  939.35   616.8  948.27   676.4  955.21   696.3  963.66
   724.1  984.88     740  990.09   775.8 1017.11   811.6 1034.28   819.5  1039.8
#Mann= 3 , 0 , 0
       0      .1       0   398.2    .045       0   420.1      .1       0
#XS Ineff= 2 , 0
       0   382.2   937.1               0
Permanent Ineff=
       F       F
Bank Sta=398.2,420.1
XS Rating Curve= 0 ,0
Exp/Cntr=0.3,0.1

Type RM Length L Ch R = 1 ,20055.5 ,495.6,500,502.3
XS GIS Cut Line= 3
     1816962.739      381693.924     1817308.871      381925.804
      1817655.44      382141.314
#Sta/Elev= 30
       0 1082.09    27.8 1069.44    43.6 1056.65    71.4 1045.82   107.1 1027.76
     123 1024.01   154.8 1007.79   226.2  957.84   253.9     929   257.9  927.04
   313.5  923.24   337.3   928.7     369  929.24   408.7  922.34   416.6  921.27
   432.5   922.2   448.3  922.33   464.2  926.61   507.8  927.42   523.6  931.57
   543.4  948.18     583  972.58   594.9  975.75   642.5 1009.57   654.4 1015.08
   670.2  1018.1   713.8 1040.68   745.5  1050.3     801 1082.44   824.7  1100.5
#Mann= 3 , 0 , 0
       0      .1       0   408.7    .045       0   432.5      .1       0
#XS Ineff= 2 , 0
       0     369  929.24               0
Permanent Ineff=
       F       F
Bank Sta=408.7,432.5
XS Rating Curve= 0 ,0
Exp/Cntr=0.3,0.1

Type RM Length L Ch R = 1 ,19555.5 ,557.7,564.1,567.9
XS GIS Cut Line= 3
     1816756.266       382051.22     1817069.248      382321.518
     1817403.443      382582.042
#Sta/Elev= 30
       0 1082.29    43.7 1053.69    47.7 1051.79    59.6 1050.45   115.3 1020.76
   139.2 1015.11   182.9  991.57   214.7  967.97   234.6  951.21   274.4  923.12
   318.1     914   326.1  915.33     334  920.37   377.8  921.48   381.7  921.07
   393.7  914.45   401.6  913.59   413.5  912.62   423.5  914.18   469.5  913.25
   489.5  921.31   509.5  917.66   541.5   921.1   621.4  986.66   641.4 1000.02
   653.4    1004   677.4 1021.65   709.4 1039.44   769.3 1067.66   837.3 1113.94
#Mann= 3 , 0 , 0
       0      .1       0   401.6    .045       0   423.5      .1       0
#XS Ineff= 2 , 0
       0   373.8   920.9               0
Permanent Ineff=
       F       F
Bank Sta=401.6,423.5
XS Rating Curve= 0 ,0
Exp/Cntr=0.3,0.1

Type RM Length L Ch R = 1 ,18991.4 ,313.1,321.8,330.3
XS GIS Cut Line= 3
     1816508.121       382422.84     1816797.183      382718.413
     1817725.511      382949.967
#Sta/Elev= 30
       0 1032.51    23.8 1024.64    55.6 1006.53    99.4  995.07     159  956.33
   214.7  910.55   246.5  904.81   266.3   912.7   294.2  912.82   310.1  905.48
     318  903.02   333.9  904.97   369.7  912.76   493.2  912.06   616.7  917.59
   668.6  915.58   708.4  919.36   744.3  929.36     836   963.8   851.9  966.67
   867.9  975.13   935.7  999.79  1043.3 1031.57  1095.1 1040.81    1127 1040.51
  1194.8 1056.78  1286.5 1074.34  1338.3 1080.16  1354.2  1087.7  1370.2 1088.01
#Mann= 3 , 0 , 0
       0      .1       0   310.1    .045       0   333.9      .1       0
#XS Ineff= 2 , 0
       0     290   912.4               0
Permanent Ineff=
       F       F
Bank Sta=310.1,333.9
XS Rating Curve= 0 ,0
Exp/Cntr=0.3,0.1

Type RM Length L Ch R = 1 ,18669.6 ,583.1,597.6,609.4
XS GIS Cut Line= 3
       1816301.9        382470.8     1816548.052      383005.306
     1817260.233      383585.384
#Sta/Elev= 30
       0 1045.38    15.9  1035.5    51.7 1026.94    87.5  1004.2   103.4 1001.08
   131.2   986.8     171   957.7   202.8  928.82   222.7  916.43   278.3  903.04
   389.7  898.04   401.6  896.78   421.5  897.84   453.3  901.26   465.2   905.6
   560.6  904.57   600.4  907.41   612.4  912.85   680.3  958.41   736.2  985.92
   804.1 1006.48   832.1 1009.27     852 1015.85     900    1026  1027.8  1038.7
  1175.5 1044.31  1235.4 1044.36  1271.4 1041.66  1363.2 1048.44    1507 1044.77
#Mann= 3 , 0 , 0
       0     .09       0   389.7    .045       0   421.5     .09       0
Bank Sta=389.7,421.5
XS Rating Curve= 0 ,0
Exp/Cntr=0.3,0.1

Type RM Length L Ch R = 1 ,18072   ,367.9,378.7,390
XS GIS Cut Line= 2
     1815953.433      382559.993     1815916.975      383362.076
#Sta/Elev= 30
       0 1021.93      12 1017.21    43.9  997.36    59.9  993.07    79.9  981.58
   107.8  958.85   131.8  944.52   147.8  932.39   167.8  921.28   187.8  899.83
   243.7  894.86   255.6  900.88   279.6  902.15   283.6  901.83   295.6  893.56
   303.6  892.08   355.5  894.06   466.7  891.51   479.4  890.68   487.3  891.55
   511.3  897.13   547.3  917.71   595.2  952.53   619.2  972.69   631.1  976.53
   651.1  991.91     703 1017.16     727 1027.26     735 1028.52   802.9 1065.68
#Mann= 3 , 0 , 0
       0      .1       0   466.7    .045       0   487.3      .1       0
#XS Ineff= 2 , 0
       0   283.6                       0
Permanent Ineff=
       F       F
Bank Sta=466.7,487.3
XS Rating Curve= 0 ,0
Exp/Cntr=0.3,0.1

Type RM Length L Ch R = 1 ,17693.3 ,235.4,236.9,238.5
XS GIS Cut Line= 2
     1815797.183      382489.681     1815469.058      383216.243
#Sta/Elev= 30
       0 1001.56      12  993.95    67.8  978.85   111.6  952.71   127.6  950.56
   147.5   938.4   163.4  925.27   187.4  916.46   223.2  896.26   247.1  893.57
   255.1  890.62     275  892.45     295  891.24   306.9  896.08   334.8  897.59
   358.8  887.66   366.7  887.37   379.2  888.03   386.6  889.76   422.5  889.19
   442.5  893.25   486.3  894.69   502.2  897.75   613.9  900.11   633.8     903
   649.7  910.01   721.5  958.13   749.4  974.73   769.3  983.48   797.2  989.42
#Mann= 3 , 0 , 0
       0      .1       0   358.8    .045       0   379.2      .1       0
#XS Ineff= 2 , 0
       0   330.8                       0
Permanent Ineff=
       F       F
Bank Sta=358.8,379.2
XS Rating Curve= 0 ,0
Exp/Cntr=0.3,0.1

Type RM Length L Ch R = 1 ,17456.3 ,139.5,129.3,118.2
XS GIS Cut Line= 2
      1815703.81      382211.035      1815241.57      383084.733
#Sta/Elev= 30
       0 1062.72       8 1055.76    27.9 1049.45    59.8  1030.7    83.7 1027.96
   135.5  998.13   167.4  986.34   211.2     953   219.2  949.02   235.2  945.45
     267  927.07     291  908.86   302.9  902.41   346.8  895.36   402.6  894.24
   418.5   890.6   442.4  891.46   474.3  887.88   494.2  888.85   510.2  895.03
     542  896.31     566   886.6   581.9  885.67   593.9  886.61   709.4  892.46
   773.2  893.63     825  898.74   860.9  894.63   900.8  902.32   988.4  907.91
#Mann= 3 , 0 , 0
       0      .1       0     566    .045       0   593.9      .1       0
#XS Ineff= 2 , 0
       0   538.1                       0
Permanent Ineff=
       F       F
Bank Sta=566,593.9
XS Rating Curve= 0 ,0
Exp/Cntr=0.3,0.1

Type RM Length L Ch R = 1 ,17327   ,78.4,78,78.4
XS GIS Cut Line= 4
      1815520.65      382129.004     1815326.205       382576.92
     1815314.053      382714.073     1815067.525      383106.434
#Sta/Elev= 30
       0  1022.9    39.7 1005.34    99.2  985.75     131  959.51   154.8  952.63
   178.6  936.37   218.4  922.35   250.1  903.55     270  895.92   313.6   892.4
   357.3  892.57   369.2  889.56   456.5  889.01   472.4  886.03   492.2  892.19
   531.6   894.5   543.4  889.08     567  885.74   570.9  885.44   586.6  885.83
     654  891.41   809.8  895.92   817.7  899.02   841.7   916.7   877.7  936.56
   893.6  939.88   905.6  948.05   945.6   964.2  1025.5  989.99  1089.4  998.16
#Mann= 3 , 0 , 0
       0      .1       0     567    .045       0   586.6     .09       0
#XS Ineff= 2 , 0
       0   527.6                       0
Permanent Ineff=
       F       F
Bank Sta=567,586.6
XS Rating Curve= 0 ,0
Exp/Cntr=0.3,0.1

Type RM Length L Ch R = 1 ,17249   ,107.7,117.8,128
XS GIS Cut Line= 4
     1815450.251      382113.986     1815255.806      382561.903
     1815243.653      382699.056     1814997.126      383091.417
#Sta/Elev= 30
       0  999.57    23.8   995.1    47.6  985.72    83.4  965.55     139  947.48
   190.6  925.69   222.3  921.22   234.2  912.17     258  900.49   313.6  896.94
   349.4  891.31   460.5  886.49   476.4  891.09     508  891.23   527.6  885.78
   547.3  884.45     567   884.2   574.8  884.41   606.3  891.51   785.8  893.84
   789.8  895.44   801.8  908.98   829.7  928.81   869.7  947.16   885.6  951.13
   897.6  959.71   965.5  990.36   993.5 1005.78  1049.4 1021.75  1089.4 1023.47
#Mann= 3 , 0 , 0
       0      .1       0   547.3    .045       0   574.8      .1       0
#XS Ineff= 2 , 0
       0     508                       0
Permanent Ineff=
       F       F
Bank Sta=547.3,574.8
XS Rating Curve= 0 ,0
Exp/Cntr=0.3,0.1

Type RM Length L Ch R = 1 ,17131.2 ,366.9,367.7,368.4
XS GIS Cut Line= 2
     1815369.174      382129.004     1814925.164       383007.91
#Sta/Elev= 30
       0   949.7       8  950.39    31.9  946.68   111.6  919.26   139.5  913.52
   167.4  912.38   195.3  908.69   219.3  903.33   271.1  897.89     291  898.07
   354.8  889.79   418.6  886.18   430.6  889.33   458.5  891.81   478.4   884.2
   491.9  883.08   506.3  882.66   514.3  883.11     598  889.18   709.6  889.51
   725.6  907.73   765.4  935.42   781.4  940.62   789.4  946.33   829.2   964.2
   841.2  971.35   869.1  976.16     885  983.92   964.8 1005.02   984.7 1012.66
#Mann= 3 , 0 , 0
       0      .1       0   491.9    .045       0   514.3      .1       0
#XS Ineff= 2 , 0
       0   458.5             620       0
Permanent Ineff=
       F       F
Bank Sta=491.9,514.3
XS Rating Curve= 0 ,0
Exp/Cntr=0.3,0.1

Type RM Length L Ch R = 1 ,16763.5 ,483.6,470.6,457.5
XS GIS Cut Line= 3
     1815017.922      382056.392     1814829.046      382419.032
      1814632.45      382782.264
#Sta/Elev= 30
       0  953.19    11.9  945.81    83.4  909.17   103.2  901.88   115.1   895.6
     135  891.14   182.6  888.54   293.8  886.45   333.4  882.31   349.3   886.9
   369.2  887.07   377.1  886.45     393  880.94   416.8  881.16   431.1   879.4
   440.6  878.73   456.5  879.43   472.4  883.41   603.5  883.67   607.4  886.06
   619.4  899.02   627.3  904.94   643.2     913   659.1  924.36   678.9  935.67
   722.6  958.64   758.4  975.75   798.1  988.61     814  992.15   821.9  995.35
#Mann= 3 , 0 , 0
       0      .1       0   431.1    .045       0   456.5      .1       0
#XS Ineff= 2 , 0
       0   361.2                       0
Permanent Ineff=
       F       F
Bank Sta=431.1,456.5
XS Rating Curve= 0 ,0
Exp/Cntr=0.3,0.1

Type RM Length L Ch R = 1 ,16292.9 ,560.5,572.1,583.8
XS GIS Cut Line= 3
       1814557.6      381872.493     1814403.954      382187.597
     1814419.579      382734.472
#Sta/Elev= 30
       0 1012.02    19.9 1006.79    35.8  997.09    55.8  980.23    71.7  957.07
    79.7  951.39   167.3  947.15   219.1  906.51     247   888.9   266.9  883.38
   318.7  876.98   334.6  881.14   374.5  884.18   390.5  875.96   402.5  874.74
   418.5  874.01   430.4  874.67   462.4  877.99   502.3   876.2   566.2  879.43
   622.1   884.8   634.1  890.24   658.1  910.09     690  907.68     702  916.51
   733.9  930.45   793.8   964.1   813.8  966.84   821.8  972.12   897.7  998.57
#Mann= 3 , 0 , 0
       0      .1       0   402.5    .045       0   430.4      .1       0
#XS Ineff= 2 , 0
       0   370.5                       0
Permanent Ineff=
       F       F
Bank Sta=402.5,430.4
XS Rating Curve= 0 ,0
Exp/Cntr=0.3,0.1

Type RM Length L Ch R = 1 ,15720.8 ,776.9,770.7,764.3
XS GIS Cut Line= 2
     1814112.288      381573.014     1813747.704      382472.319
#Sta/Elev= 30
       0 1044.41      24 1037.62    75.9 1008.78    91.8  991.06   103.8  986.23
   123.8  954.66   127.8  951.88   211.6  949.33   227.6  941.35   263.6  931.47
   339.4  878.22   403.3  872.39   415.3  876.68   443.3  876.86   459.2  869.89
   475.2   869.3   487.2  868.98   499.2   869.2   515.2  874.68     579  871.42
   686.9  872.27   714.8  900.07   750.8  924.33   778.7  939.21   846.6  966.97
   866.6  970.95   890.5  980.69   926.5 1004.25   958.4 1012.81   970.4 1020.77
#Mann= 3 , 0 , 0
       0      .1       0   475.2    .045       0   499.2      .1       0
Bank Sta=475.2,499.2
XS Rating Curve= 0 ,0
Exp/Cntr=0.3,0.1

Type RM Length L Ch R = 1 ,14950.1 ,428.6,427.1,425.9
XS GIS Cut Line= 2
     1813331.038      381152.875     1813174.788      382180.653
#Sta/Elev= 30
       0 1031.03      56 1015.95      80 1000.93      96  985.49     108  950.88
     124  943.72   147.9  940.87   175.9  945.11   199.9  944.35   223.9  935.52
   311.9  929.57   339.9  918.56   395.8  888.03   483.8  877.64   507.8  864.77
   523.8  868.32   559.8  868.56   575.8  862.02   587.8  861.39   607.8  861.19
   611.8   861.6   623.8  866.52   643.7  868.23   743.7  867.99   755.7  874.56
   779.7   894.9   799.7  905.02   919.6  951.28   987.6  969.62  1039.6  989.84
#Mann= 3 , 0 , 0
       0      .1       0   587.8    .045       0   611.8      .1       0
#XS Ineff= 2 , 0
       0                     643       0
Permanent Ineff=
       F       F
Bank Sta=587.8,611.8
XS Rating Curve= 0 ,0
Exp/Cntr=0.3,0.1

Type RM Length L Ch R = 1 ,14523.1 ,145.9,133.7,122.7
XS GIS Cut Line= 2
     1812881.327      381168.934     1812789.313      381964.073
#Sta/Elev= 30
       0  951.59    55.8  955.91    71.7   952.4   115.5   950.2   131.4  950.71
   135.4  949.36   143.4   943.1   163.3  930.66   195.1  908.26   211.1  895.22
     231  881.05   242.9  875.53   270.8  867.42   310.6  864.02   354.4  863.75
   370.4  861.54   394.2  863.62     442   864.8   485.8  856.57   501.8  858.29
   529.6   857.6   545.6  856.63   553.5  857.66   565.5  862.24   613.3  862.52
   645.1  866.75     677  879.12   720.8  905.43   760.6  923.93   800.4  935.89
#Mann= 3 , 0 , 0
       0      .1       0   529.6    .045       0   553.5      .1       0
Bank Sta=529.6,553.5
XS Rating Curve= 0 ,0
Exp/Cntr=0.3,0.1

Type RM Length L Ch R = 1 ,14389.3 ,89.6,92.3,93.1
XS GIS Cut Line= 5
     1812810.363      381105.349     1812682.325      381575.184
     1812712.477      381676.604     1812691.006      381732.519
     1812763.705      381997.276
#Sta/Elev= 30
       0  952.25       8  949.52      20  952.39    67.9  951.05    99.8  955.17
   115.8  951.82   155.7  950.66   175.6  938.32   215.5  921.67   243.5  897.36
   267.4  879.84   287.4  870.51   311.3  863.73   399.2  862.64   423.1   859.6
   443.1  862.93     471  862.34     487  859.57   514.4  861.26   545.3  855.84
   549.7  855.54   565.3  856.11   624.7     858   644.7   863.1   736.2  864.87
   744.2  868.66     780  895.78   835.7  926.64   867.5  937.95   927.2  949.44
#Mann= 3 , 0 , 0
       0      .1       0   545.3    .045       0   565.3      .1       0
Bank Sta=545.3,565.3
XS Rating Curve= 0 ,0
Exp/Cntr=0.3,0.1

Type RM Length L Ch R = 1 ,14297.1 ,97.7,106.6,112
XS GIS Cut Line= 4
     1812730.068      381132.476       1812604.2      381454.741
      1812602.03      381602.311     1812721.388      382003.787
#Sta/Elev= 30
       0  952.59    27.8  957.07    51.7  951.12   107.4  950.52   119.3  945.54
   190.9  894.42   198.8  892.54   218.7  896.36   270.4  893.52   298.2  880.82
   318.1  867.51   330.1  862.05   369.9  861.37   385.9  857.32   497.6  859.96
   513.5  859.08   525.5  854.89   541.4  854.44   549.4  854.99   573.3   857.2
   609.2  856.19   629.2  864.54   720.9  867.69   724.9  869.86   752.8  895.88
   788.7  916.47   820.7  931.38   852.6  944.41   884.5  953.08   912.4  956.02
#Mann= 3 , 0 , 0
       0      .1       0   525.5    .045       0   549.4      .1       0
Bank Sta=525.5,549.4
XS Rating Curve= 0 ,0
Exp/Cntr=0.3,0.1

Type RM Length L Ch R = 1 ,14190.5 ,277.6,289.7,305.1
XS GIS Cut Line= 3
     1812730.285      381052.615     1812506.327      381431.087
     1812579.244      382004.004
#Sta/Elev= 30
       0  980.01      28  957.34      40  952.52      80  957.85   107.9  957.44
   135.9  952.14   175.9   952.6   251.9  898.79   271.9  894.88   291.8  897.26
   347.8  871.92   459.7  878.31   499.5  854.32   563.2  851.76   599.1  859.01
     627  859.69   642.9  864.75   658.8  865.65   690.7  854.88   722.3  853.52
   742.3  853.54   754.4   856.8   766.4  864.42     854     882   905.8  903.82
   945.6  932.34   973.5  947.07   989.4     950  1005.4  947.52  1017.3  952.57
#Mann= 3 , 0 , 0
       0      .1       0   722.3    .045       0   742.3      .1       0
Bank Sta=722.3,742.3
XS Rating Curve= 0 ,0
Exp/Cntr=0.3,0.1

Type RM Length L Ch R = 1 ,13900.8 ,620.7,619.4,617.8
XS GIS Cut Line= 2
     1812742.496      380955.392     1812063.242      382023.101
#Sta/Elev= 30
       0 1022.59    39.9 1014.78    75.8 1000.73    91.8  976.99   119.8  956.04
   155.7  961.06   199.6  953.25   255.5  953.33   299.4  925.94   327.3   905.1
   367.3  900.02   423.2  865.84     511  866.46   538.9  872.54   578.8  872.66
   602.8  861.39   634.7  852.55   837.7  850.01   842.3  849.31   857.7  850.38
   878.2  856.67   942.1  863.85     970  882.69  1033.9  910.23  1085.8  943.28
  1141.7  944.86  1153.7  948.19  1181.6  966.27  1209.6  995.16  1265.5 1013.01
#Mann= 3 , 0 , 0
       0      .1       0   837.7    .045       0   857.7     .09       0
Bank Sta=837.7,857.7
XS Rating Curve= 0 ,0
Exp/Cntr=0.3,0.1

Type RM Length L Ch R = 1 ,13281.4 ,630.6,623.4,616.4
XS GIS Cut Line= 3
     1811839.718      380638.552     1811965.586      381083.431
     1811598.833      381758.344
#Sta/Elev= 30
       0 1079.51    15.9 1067.23    27.9 1065.54    47.8 1055.36    95.7 1024.21
   115.6 1021.07   179.4  991.97   203.3   963.6   219.2  951.16   255.1  946.23
   322.8  949.02   366.7  927.81   378.6  918.93   422.5  918.14   462.3  888.64
   470.3  886.19     522  881.96   561.8  874.18   701.1  866.03     737  857.69
   876.2  852.45   900.1  854.76     916  844.47     928  843.47   951.9  844.27
   983.7  845.82  1011.6   855.4  1166.8  879.18  1190.7  887.47  1230.5  914.16
#Mann= 3 , 0 , 0
       0      .1       0     916    .045       0   951.9     .09       0
#XS Ineff= 2 , 0
       0     900                       0
Permanent Ineff=
       F       F
Bank Sta=916,951.9
XS Rating Curve= 0 ,0
Exp/Cntr=0.3,0.1
